--- PNTHRCMPCK.prj (project) ---

Proj Title=PNTHRCMPCK
Current Plan=p01
Default Exp/Contr=0.3,0.1
English Units
Geom File=g01
Flow File=f01
Plan File=p01
Y Axis Title=Elevation
X Axis Title(PF)=Main Channel Distance
X Axis Title(XS)=Station
BEGIN DESCRIPTION:
Stream Name- Panther Camp Creek
Flood Zone: Zone A
Greenbrier County, WV
County-Wide Study
WVDHSEM-2018-3, Flood Risk Project
HEC-RAS Version: 5.0.7
General Notes:
For the Hydrology Regression was used.
END DESCRIPTION:
DSS Export Rating Curves= 0
DSS Export Rating Curve Sorted= 0
DSS Export Volume Flow Curves= 0
DXF Filename=A3a.
DXF OffsetX= 0
DXF OffsetY= 0
DXF ScaleX= 1
DXF ScaleY= 10

--- PNTHRCMPCK.p01 (plan) ---

Plan Title=Floodplain
Program Version=5.07
Short Identifier=Floodplain
Geom File=g01
Flow File=f01
Subcritical Flow
K Sum by GR= 0
Std Step Tol= 0.01
Critical Tol= 0.01
Num of Std Step Trials= 20
Max Error Tol= 0.3
Flow Tol Ratio= 0.001
Split Flow NTrial= 30
Split Flow Tol= 0.02
Split Flow Ratio= 0.02
Log Output Level= 0
Friction Slope Method= 1
Unsteady Friction Slope Method= 2
Unsteady Bridges Friction Slope Method= 1
Parabolic Critical Depth
Global Vel Dist= 0 , 0 , 0
Global Log Level= 0
CheckData=True
Encroach Param=-1 ,0,0, 0
Computation Interval=1MIN
Output Interval=1HOUR
Instantaneous Interval=1HOUR
Mapping Interval=1HOUR
Computation Time Step Use Courant=        0
Computation Time Step Use Time Series=    0
Computation Time Step Count To Double=0
Computation Time Step Max Doubling=0
Computation Time Step Max Halving=0
Computation Time Step Residence Courant=0
Run HTab= 0
Run UNet= 0
Run Sediment= 0
Run PostProcess= 0
Run WQNet= 0
Run RASMapper= 0
UNET Theta= 1
UNET Theta Warmup= 1
UNET ZTol= 0.02
UNET ZSATol= 0.02
UNET MxIter= 20
UNET Max Iter WO Improvement= 0
UNET MaxInSteps= 0
UNET DtIC= 0
UNET DtMin= 0
UNET MaxCRTS= 20
UNET WFStab= 2
UNET SFStab= 1
UNET WFX= 1
UNET SFX= 1
UNET 1D Methodology=Finite Difference
UNET DSS MLevel= 4
UNET Pardiso=0
UNET DZMax Abort= 100
UNET Use Existing IB Tables=-1
UNET Froude Reduction=False
UNET Froude Limit= 0.8
UNET Froude Power= 4
UNET D1 Cores= 0
UNET D2 Coriolis=0
UNET D2 Cores= 0
UNET D2 Theta= 1
UNET D2 Theta Warmup= 1
UNET D2 Z Tol= 0.01
UNET D2 Volume Tol= 0.01
UNET D2 Max Iterations= 20
UNET D2 Equation= 0
UNET D2 RampUpFraction=0.1
UNET D2 TimeSlices= 1
UNET D2 BCVolumeCheck=0
UNET D1D2 MaxIter= 0
UNET D1D2 ZTol=0.01
UNET D1D2 QTol=0.1
UNET D1D2 MinQTol=1
Write IC File= 0
Write IC File at Fixed DateTime=0
Write IC File at Sim End=0
Echo Input=False
Echo Parameters=False
Echo Output=False
Write Detailed= 0
HDF Write Warmup=0
HDF Write Time Slices=0
HDF Flush=0
HDF Face Node Velocities=0
HDF Compression= 1
HDF Chunk Size= 1
HDF Spatial Parts= 1
HDF Use Max Rows=0
HDF Fixed Rows= 1
Calibration Method= 0
Calibration Iterations= 20
Calibration Max Change=0.05
Calibration Tolerance=0.2
Calibration Maximum=1.5
Calibration Minimum=0.5
Calibration Optimization Method= 1
WQ AD Non Conservative
WQ ULTIMATE=-1
WQ Max Comp Step=1HOUR
WQ Output Interval=15MIN
WQ Output Selected Increments= 0
WQ Output face flow=0
WQ Output face velocity=0
WQ Output face area=0
WQ Output face dispersion=0
WQ Output cell volume=0
WQ Output cell surface area=0
WQ Output cell continuity=0
WQ Output cumulative cell continuity=0
WQ Output face conc=0
WQ Output face dconc_dx=0
WQ Output face courant=0
WQ Output face peclet=0
WQ Output face adv mass=0
WQ Output face disp mass=0
WQ Output cell mass=0
WQ Output cell source sink temp=0
WQ Output nsm pathways=0
WQ Output nsm derived pathways=0
WQ Output MaxMinRange=-1
WQ Daily Max Min Mean=-1
WQ Daily Range=0
WQ Daily Time=0
WQ Create Restart=0
WQ Fixed Restart=0
WQ System Summary=0
WQ Write To DSS=0
WQ Use Fixed Temperature=0
Sorting and Armoring Iterations= 10
XS Update Threshold= 0.02
Bed Roughness Predictor= 0
Hydraulics Update Threshold= 0.02
Energy Slope Method= 1
Volume Change Method= 1
Sediment Retention Method= 0
XS Weighting Method= 0
Number of US Weighted Cross Sections= 1
Number of DS Weighted Cross Sections= 1
Upstream XS Weight=0
Main XS Weight=1
Downstream XS Weight=0
Number of DS XS's Weighted with US Boundary= 1
Upstream Boundary Weight= 1
Weight of XSs Associated with US Boundary= 0
Number of US XS's Weighted with DS Boundary= 1
Downstream Boundary Weight= 0.5
Weight of XSs Associated with DS Boundary= 0.5
Percentile Method= 0
Sediment Output Level= 3
Mass or Volume Output= 0
Output Increment Type= 1
Profile and TS Output Increment= 1
XS Output Flag= 0
XS Output Increment= 10
Write Gradation File= 0
Read Gradation Hotstart= 0
Write HDF5 File= 1
Write Binary Output= 1
Write DSS Sediment File= 0
SV Curve= 0
Specific Gage Flag= 0

--- PNTHRCMPCK.f01 (steady flow) ---

Flow Title=Flow
Program Version=5.07
Number of Profiles= 6
Profile Names=f1p,f10p,f4p,f2p,f02p,f1pplus
River Rch & RM=BEVERLYFK,Main            ,776
     323     167     225     272     456     478
River Rch & RM=BEVERLYFK,Main            ,220
     537     283     377     454     751     794
River Rch & RM=BOGGSRN,Main            ,1733
     558     295     392     472     780     825
River Rch & RM=DRYRN,Main            ,9301
     532     280     373     450     744     787
River Rch & RM=DRYRN,Main            ,8316
     594     314     418     503     829     878
River Rch & RM=DRYRN,Main            ,6862
     769     411     544     653    1070    1140
River Rch & RM=DRYRN,Main            ,5213
     898     483     637     763    1240    1330
River Rch & RM=DRYRN,Main            ,259
    1110     604     793     948    1540    1650
River Rch & RM=PNTHRCMPCK,Main            ,14558
     513     270     359     434     718     758
River Rch & RM=PNTHRCMPCK,Main            ,13060
     599     317     422     508     836     886
River Rch & RM=PNTHRCMPCK,Main            ,10150
     873     469     619     742    1210    1290
River Rch & RM=PNTHRCMPCK,Main            ,8160
     976     526     693     830    1350    1440
River Rch & RM=PNTHRCMPCK,Main            ,6420
    1080     588     772     923    1500    1600
River Rch & RM=RCKCMPRN,Main            ,4355
     581     307     409     492     812     860
River Rch & RM=RCKCMPRN,Main            ,1618
     692     368     488     586     963    1020
River Rch & RM=ROBBINSRN,Main            ,27789
     907     488     643     771    1260    1340
River Rch & RM=ROBBINSRN,Main            ,27014
    1170     638     837    1000    1620    1740
River Rch & RM=ROBBINSRN,Main            ,21785
    1330     728     953    1140    1830    1970
River Rch & RM=ROBBINSRN,Main            ,16781
    1830    1010    1320    1570    2500    2710
River Rch & RM=ROBBINSRN,Main            ,10962
    2050    1140    1480    1750    2790    3030
River Rch & RM=SPRINGCKT3,Main            ,6529
     583     309     410     494     815     863
River Rch & RM=SPRINGCKT3,Main            ,3093
     683     363     482     579     951    1010
River Rch & RM=SPRINGCKT3,Main            ,434
     860     462     609     730    1190    1270
Boundary for River Rch & Prof#=BEVERLYFK,Main            , 1
Up Type= 0
Dn Type= 3
Dn Slope=0.045649
Boundary for River Rch & Prof#=BEVERLYFK,Main            , 2
Up Type= 0
Dn Type= 3
Dn Slope=0.045649
Boundary for River Rch & Prof#=BEVERLYFK,Main            , 3
Up Type= 0
Dn Type= 3
Dn Slope=0.045649
Boundary for River Rch & Prof#=BEVERLYFK,Main            , 4
Up Type= 0
Dn Type= 3
Dn Slope=0.045649
Boundary for River Rch & Prof#=BEVERLYFK,Main            , 5
Up Type= 0
Dn Type= 3
Dn Slope=0.045649
Boundary for River Rch & Prof#=BEVERLYFK,Main            , 6
Up Type= 0
Dn Type= 3
Dn Slope=0.045649
Boundary for River Rch & Prof#=BOGGSRN,Main            , 1
Up Type= 0
Dn Type= 3
Dn Slope=0.043074
Boundary for River Rch & Prof#=BOGGSRN,Main            , 2
Up Type= 0
Dn Type= 3
Dn Slope=0.043074
Boundary for River Rch & Prof#=BOGGSRN,Main            , 3
Up Type= 0
Dn Type= 3
Dn Slope=0.043074
Boundary for River Rch & Prof#=BOGGSRN,Main            , 4
Up Type= 0
Dn Type= 3
Dn Slope=0.043074
Boundary for River Rch & Prof#=BOGGSRN,Main            , 5
Up Type= 0
Dn Type= 3
Dn Slope=0.043074
Boundary for River Rch & Prof#=BOGGSRN,Main            , 6
Up Type= 0
Dn Type= 3
Dn Slope=0.043074
Boundary for River Rch & Prof#=DRYRN,Main            , 1
Up Type= 0
Dn Type= 3
Dn Slope=0.021282
Boundary for River Rch & Prof#=DRYRN,Main            , 2
Up Type= 0
Dn Type= 3
Dn Slope=0.021282
Boundary for River Rch & Prof#=DRYRN,Main            , 3
Up Type= 0
Dn Type= 3
Dn Slope=0.021282
Boundary for River Rch & Prof#=DRYRN,Main            , 4
Up Type= 0
Dn Type= 3
Dn Slope=0.021282
Boundary for River Rch & Prof#=DRYRN,Main            , 5
Up Type= 0
Dn Type= 3
Dn Slope=0.021282
Boundary for River Rch & Prof#=DRYRN,Main            , 6
Up Type= 0
Dn Type= 3
Dn Slope=0.021282
Boundary for River Rch & Prof#=PNTHRCMPCK,Main            , 1
Up Type= 0
Dn Type= 3
Dn Slope=0.02712
Boundary for River Rch & Prof#=PNTHRCMPCK,Main            , 2
Up Type= 0
Dn Type= 3
Dn Slope=0.02712
Boundary for River Rch & Prof#=PNTHRCMPCK,Main            , 3
Up Type= 0
Dn Type= 3
Dn Slope=0.02712
Boundary for River Rch & Prof#=PNTHRCMPCK,Main            , 4
Up Type= 0
Dn Type= 3
Dn Slope=0.02712
Boundary for River Rch & Prof#=PNTHRCMPCK,Main            , 5
Up Type= 0
Dn Type= 3
Dn Slope=0.02712
Boundary for River Rch & Prof#=PNTHRCMPCK,Main            , 6
Up Type= 0
Dn Type= 3
Dn Slope=0.02712
Boundary for River Rch & Prof#=RCKCMPRN,Main            , 1
Up Type= 0
Dn Type= 3
Dn Slope=0.013802
Boundary for River Rch & Prof#=RCKCMPRN,Main            , 2
Up Type= 0
Dn Type= 3
Dn Slope=0.013802
Boundary for River Rch & Prof#=RCKCMPRN,Main            , 3
Up Type= 0
Dn Type= 3
Dn Slope=0.013802
Boundary for River Rch & Prof#=RCKCMPRN,Main            , 4
Up Type= 0
Dn Type= 3
Dn Slope=0.013802
Boundary for River Rch & Prof#=RCKCMPRN,Main            , 5
Up Type= 0
Dn Type= 3
Dn Slope=0.013802
Boundary for River Rch & Prof#=RCKCMPRN,Main            , 6
Up Type= 0
Dn Type= 3
Dn Slope=0.013802
Boundary for River Rch & Prof#=ROBBINSRN,Main            , 1
Up Type= 0
Dn Type= 3
Dn Slope=0.010317
Boundary for River Rch & Prof#=ROBBINSRN,Main            , 2
Up Type= 0
Dn Type= 3
Dn Slope=0.010317
Boundary for River Rch & Prof#=ROBBINSRN,Main            , 3
Up Type= 0
Dn Type= 3
Dn Slope=0.010317
Boundary for River Rch & Prof#=ROBBINSRN,Main            , 4
Up Type= 0
Dn Type= 3
Dn Slope=0.010317
Boundary for River Rch & Prof#=ROBBINSRN,Main            , 5
Up Type= 0
Dn Type= 3
Dn Slope=0.010317
Boundary for River Rch & Prof#=ROBBINSRN,Main            , 6
Up Type= 0
Dn Type= 3
Dn Slope=0.010317
Boundary for River Rch & Prof#=SPRINGCKT3,Main            , 1
Up Type= 0
Dn Type= 3
Dn Slope=0.016207
Boundary for River Rch & Prof#=SPRINGCKT3,Main            , 2
Up Type= 0
Dn Type= 3
Dn Slope=0.016207
Boundary for River Rch & Prof#=SPRINGCKT3,Main            , 3
Up Type= 0
Dn Type= 3
Dn Slope=0.016207
Boundary for River Rch & Prof#=SPRINGCKT3,Main            , 4
Up Type= 0
Dn Type= 3
Dn Slope=0.016207
Boundary for River Rch & Prof#=SPRINGCKT3,Main            , 5
Up Type= 0
Dn Type= 3
Dn Slope=0.016207
Boundary for River Rch & Prof#=SPRINGCKT3,Main            , 6
Up Type= 0
Dn Type= 3
Dn Slope=0.016207
DSS Import GetInterval= 0
DSS Import GetPeak= 0
DSS Import FillOption= 0

--- PNTHRCMPCK.g01 (geometry) ---

Geom Title=Geometry
Program Version=5.07

River Reach=PNTHRCMPCK      ,Main
Reach XY= 30
2141046.81985147405985.1300213042140554.26014106405563.010130644
2140514.37997147405241.0301315642140276.11010681405158.920059562
2140185.92984097404573.7099438912139877.25985464403896.759854227
2139931.68002139403433.1098628942139673.77010414403087.450121149
2139789.17997831402989.6599624012140050.93011098402010.960148141
2140247.91987447401709.9801070542140009.25991872401276.770015478
2139989.29014239400977.430062979 2140114.7600358400801.740125641
2140102.40015239400531.7400094722140344.31994414399707.510030642
2140582.16986214 399483.350045892140440.61010589398500.870055482
2140195.37995331398301.2398773132140135.65992838398113.049964979
 2140300.2399798397676.9399448042140636.34987189 397531.10001339
2140712.60004747397280.8200021392140437.74003288396313.739915311
2140619.67995772395840.1299701482140538.43012021395397.769962475
2140630.80001423395269.3000750542140610.65996264394567.209943816
2140834.96003897394089.4300594782141412.29156147393800.840085477

Type RM Length L Ch R = 1 ,14558   ,184.8,182.9,178
XS GIS Cut Line= 2
2141453.52343439405780.3961788122140639.72158431406177.531867474
#Sta/Elev= 30
       0 2872.91    23.6  2865.7    52.4 2849.57    67.4 2845.36      99 2831.32
   123.6 2822.89   180.6 2797.99   195.2 2793.82   226.6 2780.95     239 2774.18
   290.4 2761.11   343.4 2753.88   388.3 2740.79   436.1 2705.35  447.862690.194
   455.6 2688.72  477.282690.392     493 2697.75   538.3 2698.34   567.3 2716.09
   611.3 2752.88   629.6 2763.57   728.2 2789.49   750.1 2796.76   790.9  2803.8
   812.1 2813.31   852.3 2824.99   869.4 2833.78   893.9 2851.33   905.5 2850.87
#Mann= 3 ,-1 , 0
       0      .1       0  447.86    .045       0  477.28      .1       0
Bank Sta=447.86,477.28
XS Rating Curve= 0 ,0
Exp/Cntr=0.3,0.1

Type RM Length L Ch R = 1 ,14375   ,293.1,294.1,294.6
XS GIS Cut Line= 3
2141243.02024648405564.4674768152140878.43665805405887.818208054
2140587.63802706406153.660196066
#Sta/Elev= 30
       0 2866.36    71.5 2838.22   160.4 2789.33   295.3 2740.36   323.1 2723.95
   352.1 2699.26   365.3 2693.47   381.2 2690.02  394.732681.875   404.4 2680.97
  415.452681.224   422.3 2682.53   434.6 2689.23   448.6 2692.36   479.3 2717.94
   528.1 2746.25   560.1 2755.65   643.7 2769.15   671.6  2775.8   706.4 2790.24
   736.6 2807.95     777 2835.56   808.1 2847.21   825.9 2851.54   841.1 2859.81
   852.6 2860.59     862 2853.69   865.9 2853.15   871.3 2853.87   881.3 2859.58
#Mann= 3 ,-1 , 0
       0      .1       0  394.73    .045       0  415.45      .1       0
Bank Sta=394.73,415.45
XS Rating Curve= 0 ,0
Exp/Cntr=0.3,0.1

Type RM Length L Ch R = 1 ,14081   ,360,365.9,370.6
XS GIS Cut Line= 3
2141099.42670164405381.8694168032140776.44014288 405628.48670572
2140343.49743922405951.837436974
#Sta/Elev= 30
       0  2860.9    55.9 2836.27    68.2 2833.57    86.4 2824.27   140.2 2802.66
   180.4 2782.46   308.7 2737.21     348 2725.11   390.2 2703.95   410.8 2697.76
   480.4 2688.45   500.9 2676.45  519.91 2671.61   533.6 2670.03  540.24 2670.85
     550 2676.16   564.1 2677.37   577.5 2681.86     591 2689.85   623.8 2714.39
   660.2 2730.76   758.9 2768.24   803.9 2787.19   816.2 2790.27   853.1 2807.84
   873.6 2813.81   884.5  2819.4     897 2821.83   910.4 2829.32   946.7 2844.67
#Mann= 3 ,-1 , 0
       0      .1       0  519.91    .045       0  540.24      .1       0
Bank Sta=519.91,540.24
XS Rating Curve= 0 ,0
Exp/Cntr=0.3,0.1

Type RM Length L Ch R = 1 ,13715   ,411.7,409.6,405.5
XS GIS Cut Line= 3
2141079.17477363405327.922346234 2140379.3047823405409.302432805
2140032.08270772405620.891248479
#Sta/Elev= 30
       0 2858.47    23.2 2850.46    34.2 2848.75    77.2 2828.82   232.4 2769.43
   312.2 2746.69   404.1 2724.57   417.4 2717.94   447.1 2694.47   460.3 2680.36
   483.4 2661.49   512.4 2660.79  517.762658.675   527.2 2657.11  537.792657.679
   562.7 2660.65   572.6 2664.61   605.6 2664.96   628.7    2671   668.4 2673.61
   684.9 2677.07   716.6  2690.7   754.7 2701.43   795.4 2716.24   895.7 2745.44
   931.6 2758.85   943.4 2759.72  1060.4 2810.02  1092.8 2821.65  1111.2 2831.81
#Mann= 3 ,-1 , 0
       0      .1       0  517.76    .045       0  537.79      .1       0
#XS Ineff= 2 , 0
          509.82 2666.19
Permanent Ineff=
       F       F
Bank Sta=517.76,537.79
XS Rating Curve= 0 ,0
Exp/Cntr=0.3,0.1

Type RM Length L Ch R = 1 ,13305   ,241.3,245,247.3
XS GIS Cut Line= 3
2140727.61215656404977.4450288122140234.99043839405181.438059136
2139828.08967739405412.557675645
#Sta/Elev= 30
       0 2767.84    91.3 2746.11    99.8 2742.67   152.8 2730.67   180.4 2722.59
   252.8 2707.17   288.5 2701.36     306 2696.65   322.8 2689.89   331.4  2684.8
   363.7 2661.04   374.2 2651.89   380.7  2649.3   419.7    2643     434 2644.76
  475.812641.804   487.2 2639.71  494.982642.051   522.7 2672.06   528.6 2676.41
   578.7 2690.04   601.3 2692.54   623.9 2700.66   646.6 2704.31   678.1 2712.68
   710.7 2724.76   779.9 2753.15     802 2763.76   854.1 2784.17  1001.1 2830.98
#Mann= 3 ,-1 , 0
       0      .1       0  475.81    .045       0  494.98      .1       0
#XS Ineff= 2 , 0
          435.15  2647.7
Permanent Ineff=
       F       F
Bank Sta=475.81,494.98
XS Rating Curve= 0 ,0
Exp/Cntr=0.3,0.1

Type RM Length L Ch R = 1 ,13060   ,259.5,261.3,255.6
XS GIS Cut Line= 3
2140696.14502789404894.9796425552140156.86559464404927.531742811
2139707.64667681405017.592586309
#Sta/Elev= 30
       0  2771.7    51.3 2756.74      71 2752.66    97.4 2742.71   140.1 2734.39
   179.5 2723.06   215.7 2716.44   249.2 2707.17     265 2706.06   314.3 2693.06
   327.4 2686.66   347.1 2673.34   360.8 2668.66   379.4 2656.75   389.9 2646.56
   399.7  2641.2   409.6 2638.87  415.842633.112   422.7 2631.59  442.032632.821
     495 2633.39   511.5 2640.48   534.5 2647.37   564.5 2644.08   584.6 2645.67
   631.4 2662.12   651.5 2660.62   715.1 2673.44   915.8 2729.19   998.4 2759.61
#Mann= 3 ,-1 , 0
       0      .1       0  415.84    .045       0  442.03      .1       0
Bank Sta=415.84,442.03
XS Rating Curve= 0 ,0
Exp/Cntr=0.3,0.1

Type RM Length L Ch R = 1 ,12799   ,350.5,348.4,344.5
XS GIS Cut Line= 3
2140696.14502789 404704.00725548 2140067.8900508404720.283469647
2139600.22497563404814.684527561
#Sta/Elev= 30
       0 2810.49    74.2 2778.36   162.8 2745.66   225.8 2720.11   326.9 2690.79
   342.4 2689.87   356.5 2684.75   369.4  2678.1     389 2663.44   431.9 2636.62
   448.4 2633.68   454.9 2629.52   500.9 2622.67   542.82622.434   553.4 2621.36
   562.8 2622.46   576.3 2629.26   605.9 2629.89   645.6 2654.14   673.4 2656.18
   695.8 2653.29   719.2 2656.76   809.6 2682.91   866.5 2702.62   913.4  2716.5
   949.1 2730.92   963.6 2733.43     997 2748.25  1023.1 2757.47  1105.6 2800.92
#Mann= 3 ,-1 , 0
       0      .1       0   542.8    .045       0   562.8      .1       0
Bank Sta=542.8,562.8
XS Rating Curve= 0 ,0
Exp/Cntr=0.3,0.1

Type RM Length L Ch R = 1 ,12450   ,371.6,375,375.7
XS GIS Cut Line= 3
2140588.72332673 404253.703694152140011.46627913404452.271210387
2139555.73720372 404602.01074031
#Sta/Elev= 30
       0 2816.59    33.8 2798.73   116.5 2763.14   143.6 2747.93   173.9 2739.47
   228.5 2717.44     292 2694.07   346.5 2676.84   379.8  2663.3   391.6 2661.92
   446.9 2645.87   466.4 2637.43   495.9 2617.11  551.692608.624   561.6 2606.65
  574.052609.309   634.4 2615.95   679.7 2636.63   741.4 2647.95   762.9 2657.39
   782.9 2670.27   793.2 2672.86   820.8 2692.11   903.7 2739.85   916.2 2741.68
   924.4 2747.95   972.8 2769.53  1003.9 2780.89  1031.5 2787.32  1090.2 2794.62
#Mann= 3 ,-1 , 0
       0      .1       0  551.69    .045       0  574.05      .1       0
Bank Sta=551.69,574.05
XS Rating Curve= 0 ,0
Exp/Cntr=0.3,0.1

Type RM Length L Ch R = 1 ,12075   ,276.4,278,279
XS GIS Cut Line= 3
2140476.96108305404021.4987779712139915.98024964404109.389350221
2139413.59313105404205.960679397
#Sta/Elev= 30
       0 2805.74    29.2 2793.49    72.4 2770.59   140.2  2741.8   188.6 2714.13
   268.3 2676.51     358 2644.24   374.6 2642.92   407.2 2630.91   447.4 2611.48
   480.9 2603.46   504.1 2602.14  524.082594.225     534 2592.87  544.212594.531
   557.3 2598.88     614  2601.6   650.7 2622.41   677.2 2633.08   710.9 2639.16
   744.3 2637.39   811.1 2656.89   848.2 2680.49     928 2723.11   944.7 2736.24
   958.1  2739.2   974.8 2753.04   994.9 2760.29  1004.5 2769.09  1079.4 2815.14
#Mann= 3 ,-1 , 0
       0      .1       0  524.08    .045       0  544.21      .1       0
Bank Sta=524.08,544.21
XS Rating Curve= 0 ,0
Exp/Cntr=0.3,0.1

Type RM Length L Ch R = 1 ,11797   ,352.9,352.6,352.3
XS GIS Cut Line= 2
2140467.19535455403827.2711480562139326.78753039403856.568333566
#Sta/Elev= 30
       0 2798.57    32.3 2783.04    51.9 2776.34    65.1 2767.76    78.2 2765.21
   219.3 2696.56   265.7  2678.2     285 2675.72   452.3 2621.45   478.6 2605.12
     495 2590.37   573.8 2588.24  584.612582.746   590.2 2581.87  604.842583.256
   616.4 2591.91   662.4 2603.66   691.9 2622.46   708.3 2630.28   744.4 2636.66
   790.4 2640.96   872.4 2655.66   924.9 2662.07     952 2668.51   987.3 2681.98
    1030  2704.3  1049.6 2719.51  1062.8 2721.92  1072.6 2729.78  1140.8 2767.33
#Mann= 3 ,-1 , 0
       0      .1       0  584.61    .045       0  604.84      .1       0
Bank Sta=584.61,604.84
XS Rating Curve= 0 ,0
Exp/Cntr=0.3,0.1

Type RM Length L Ch R = 1 ,11445   ,236.4,232.2,228.2
XS GIS Cut Line= 3
2140432.47331114403450.7522160562139880.17290655403514.771444976
2139385.38124523403583.130560234
#Sta/Elev= 30
       0 2795.11    73.5 2758.88    80.6 2753.14    99.9 2748.38   142.8 2719.17
   181.2 2698.89   288.2 2653.21   304.7  2641.1   321.2 2640.25   360.8  2615.5
   413.7 2592.55   440.1  2575.1  487.932568.852   499.5 2567.28  505.362569.265
   519.3 2579.47   535.9 2581.73   548.2 2591.06   578.9 2604.64   642.2  2620.3
     665 2624.63     771 2632.55   826.7 2649.37   873.6 2654.08   926.8 2668.91
   956.4 2679.51   989.6 2697.92  1002.3 2700.49    1026 2715.32  1055.5 2726.63
#Mann= 3 ,-1 , 0
       0      .1       0  487.93    .045       0  505.36      .1       0
Bank Sta=487.93,505.36
XS Rating Curve= 0 ,0
Exp/Cntr=0.3,0.1

Type RM Length L Ch R = 1 ,11213   ,180.7,193.2,201.2
XS GIS Cut Line= 4
2140312.03063864403181.6549852342139934.42640696 403245.67421414
2139731.51834822403378.0525583182139360.42460223403452.922487304
#Sta/Elev= 30
       0 2751.78    35.7 2727.88    78.3 2707.79   161.5 2673.67   201.4 2660.44
   251.4  2639.2   321.2 2616.06   331.2 2610.34   347.9  2607.8   377.8 2596.95
   404.3 2584.83   451.3 2567.85  480.792561.025   490.5 2560.75  501.662561.199
   555.9 2562.82   615.1 2591.02   664.1 2602.16   693.9 2611.47   744.4 2608.06
   780.5 2618.21   794.6 2618.22   833.4 2632.57   844.8 2633.66   874.6 2648.07
   908.4 2672.31   968.6 2704.99     982 2714.66   995.4 2717.18  1003.8 2723.06
#Mann= 3 ,-1 , 0
       0      .1       0  480.79    .045       0  501.66      .1       0
Bank Sta=480.79,501.66
XS Rating Curve= 0 ,0
Exp/Cntr=0.3,0.1

Type RM Length L Ch R = 1 ,11019   ,287.3,297,299.6
XS GIS Cut Line= 2
 2140293.5844813403130.6567276422139259.51305863403250.014428556
#Sta/Elev= 30
       0 2749.01     7.3 2745.12    16.2 2737.04    39.3  2723.5   128.5 2685.68
   336.6 2605.54   376.2 2595.06   425.7  2574.5   448.9 2571.38   504.7 2568.23
   516.5 2557.79   524.8 2554.56   541.3 2557.27   577.7 2558.23   590.6 2555.49
   607.4 2554.14   623.1 2555.26   640.4 2568.52   663.5 2578.62   693.3 2579.76
   762.6 2593.17   791.9 2606.41   805.5 2615.52   821.5 2618.56   868.3 2640.85
   921.1 2656.26   944.3 2661.03   957.2 2668.23  1010.3 2690.99  1040.9 2707.92
#Mann= 3 , 0 , 0
       0      .1       0   590.6    .045       0   623.1      .1       0
Bank Sta=590.6,623.1
XS Rating Curve= 0 ,0
Exp/Cntr=0.3,0.1

Type RM Length L Ch R = 1 ,10722   ,212,214.4,216.4
XS GIS Cut Line= 4
2140287.07399563403069.8927415612139836.77010623402984.172440559
2139713.07219088402970.0664976392139399.48718813402953.790283471
#Sta/Elev= 30
       0 2753.09    13.1  2746.3    23.1 2744.06    79.9 2715.54     130  2697.2
   153.4 2685.79   290.3 2637.57   310.4 2632.91   393.8 2603.82   400.5 2600.55
   410.5 2592.16   420.6 2589.67   440.6 2578.21   450.6 2568.38   463.9 2564.49
   483.7 2544.63  493.492540.371   500.2 2539.95  513.492541.429     530 2541.43
   553.1 2546.71   566.5 2555.79   582.8 2561.08   602.5 2557.69   643.4 2559.36
   655.1 2560.79   684.6 2569.39   697.8 2567.94   793.1 2580.08   896.9  2589.6
#Mann= 3 ,-1 , 0
       0      .1       0  493.49    .045       0  513.49      .1       0
Bank Sta=493.49,513.49
XS Rating Curve= 0 ,0
Exp/Cntr=0.3,0.1

Type RM Length L Ch R = 1 ,10508   ,185.1,184,184.8
XS GIS Cut Line= 3
2140284.90372439402933.1741829812139688.11554788402725.925909817
2139380.56102534402625.428735586
#Sta/Elev= 30
       0 2739.73      22 2727.02    32.2 2724.21   127.7 2676.52   138.4 2674.01
   163.8 2662.07   194.7 2644.17   246.3 2623.38   264.9 2612.75   292.7 2602.09
   341.6 2577.76   377.7 2563.15   452.4 2537.96   469.8 2536.66   478.3  2538.4
   494.1 2531.94  514.542531.483   514.9 2531.48   528.8 2538.47   535.8 2539.65
   577.4 2536.37   589.1 2542.69   615.7 2546.97   632.9 2553.75   650.3 2551.68
     671 2545.53   750.4 2543.06   878.1 2568.02   905.7 2578.84   955.3 2581.27
#Mann= 3 ,-1 , 0
       0      .1       0   494.1    .045       0  514.54      .1       0
Bank Sta=494.1,514.54
XS Rating Curve= 0 ,0
Exp/Cntr=0.3,0.1

Type RM Length L Ch R = 1 ,10324   ,155.9,173.7,187.8
XS GIS Cut Line= 3
2140317.46340321402847.9872423022139971.27437564402637.047691455
2139450.12960296402452.165379243
#Sta/Elev= 30
       0 2720.95      37 2704.57    89.1  2675.9   104.5 2670.82     191 2629.12
   298.2 2581.87   354.5 2563.05   396.4 2534.74   411.2 2530.57     446  2529.2
   462.9 2525.12   477.4 2523.77  485.422524.873   491.3 2531.77   497.1 2532.41
   545.9  2531.3   561.3  2526.7   581.9 2528.52   588.8 2531.73   611.5 2551.05
   644.4  2563.3   687.2 2561.31   755.8 2566.19   800.3 2565.24   811.5 2571.17
   825.5 2573.79   861.9  2597.8   874.8 2602.62   916.1 2626.85   958.4 2642.11
#Mann= 3 ,-1 , 0
       0      .1       0   462.9    .045       0  485.42      .1       0
#XS Ineff= 2 , 0
                          496.89         2539.89
Permanent Ineff=
       F       F
Bank Sta=462.9,485.42
XS Rating Curve= 0 ,0
Exp/Cntr(USF)=0,0
Exp/Cntr=0.5,0.3

Type RM Length L Ch R = 1 ,10150   ,48.6,43.9,53.2
XS GIS Cut Line= 6
2140344.60015602402833.2835147872139984.78691511402571.966635915
2139961.67042198402523.7235198152139944.58431836402362.913132817
 2139877.2449688402327.7358606612139495.32029968402192.052096632
#Sta/Elev= 30
       0 2725.38    47.6 2700.35    58.6 2697.15      87  2680.9     104 2675.22
   195.6 2630.58   281.7    2599   324.8 2577.34   338.4 2573.81   362.7 2553.45
   391.1  2534.6     401 2530.62   411.4 2528.06   469.2 2525.02   522.8 2524.86
   554.6  2518.3   572.3 2517.16   589.82517.169   631.7 2521.31   684.1 2522.06
   698.9 2526.65   777.7 2527.01   795.2  2529.6   840.5 2543.76   875.4 2544.29
   920.7  2552.4     952 2555.81    1074 2618.21  1105.4 2629.98  1141.2 2647.54
#Mann= 3 ,-1 , 0
       0      .1       0   554.6    .045       0   589.8      .1       0
#XS Ineff= 3 ,-1
       0   534.6  2521.5   609.8  634.29  2521.5  634.29     750 2526.11
Permanent Ineff=
       F       F       F
Bank Sta=554.6,589.8
XS Rating Curve= 0 ,0
Exp/Cntr(USF)=0,0
Exp/Cntr=0.5,0.3

Type RM Length L Ch R = 1 ,10106   ,301.6,286.5,255.2
XS GIS Cut Line= 5
2140361.68625963402814.1872813312139997.85275905402553.875467378
2139977.75146068402389.0448207042139965.69068165 402336.78144493
2139513.41146822402157.879889394
#Sta/Elev= 30
       0 2723.71    55.1 2694.99    65.1 2691.92    79.3 2684.31   101.5 2677.39
   201.4 2631.61   257.9 2610.93   295.5 2592.06   337.5 2576.65   357.7 2563.35
   384.9 2539.19     398 2531.06   413.1 2528.13   441.3 2527.18   472.7 2521.98
   495.8 2523.34   575.22517.793   607.7 2516.36   616.8 2518.15   685.9 2521.28
   709.3 2520.31   726.3 2525.73   769.3 2525.53     823 2528.65   862.9 2535.26
   899.8 2547.19   942.1 2549.24   977.4 2553.88  1072.7 2597.86  1153.4 2640.24
#Mann= 3 ,-1 , 0
       0      .1       0   575.2    .045       0   616.8      .1       0
#XS Ineff= 2 , 0
                          687.81         2524.93
Permanent Ineff=
       F       F
Bank Sta=575.2,616.8
XS Rating Curve= 0 ,0
Exp/Cntr(USF)=0,0
Exp/Cntr=0.5,0.3

Type RM Length L Ch R = 1 ,9820    ,363.3,367.9,370
XS GIS Cut Line= 2
2140440.06876838 402167.115019562139479.78230314402115.031790391
#Sta/Elev= 30
       0 2656.17    77.4  2645.6    97.1  2640.1   133.3  2626.9   146.4 2617.78
   166.1 2609.83   251.6 2569.74     291 2553.36   304.1 2549.76   320.5 2541.55
   346.8 2525.49   369.8 2514.45  389.262510.956   396.1 2509.22  412.242510.979
   438.8 2509.32   458.5 2512.93   478.3 2513.18     503 2517.46   530.8 2516.59
   576.8 2518.29   622.8 2522.25     636 2525.61   665.5 2537.64   754.3 2554.01
   810.1 2578.17   899.1 2624.39   938.3 2645.83   951.4 2655.16   961.7 2657.84
#Mann= 4 ,-1 , 0
       0      .1       0  389.26    .045       0  412.24      .1       0
  713.56      .1       0
#XS Ineff= 2 , 0
                          460.84         2516.57
Permanent Ineff=
       F       F
Bank Sta=389.26,412.24
XS Rating Curve= 0 ,0
Exp/Cntr=0.3,0.1

Type RM Length L Ch R = 1 ,9452    ,414.8,410,404.2
XS GIS Cut Line= 3
2140468.28065422401924.0594033152140122.14322314401810.127216473
2139583.94876146401640.856229559
#Sta/Elev= 30
       0 2625.15   134.7  2567.3   169.8 2554.27   218.2 2538.24   256.9  2511.5
   264.7 2505.49     270 2500.06  274.362497.298   290.7 2496.46  294.422496.601
   321.8 2500.56   366.7 2500.93   407.7 2507.24     434 2506.52   459.5 2510.04
   511.1 2512.95   559.3 2512.95   640.7 2523.25   661.7 2528.02     680 2533.84
   693.4 2545.68   734.9 2576.71   775.9 2601.92     800 2611.93     816 2616.46
     831 2618.26   848.2  2616.6     855 2618.01   881.4 2636.66   928.6 2660.02
#Mann= 7 ,-1 , 0
       0      .1       0  209.63      .1       0  274.36    .045       0
  294.42      .1       0  348.67     .12       0  542.18      .1       0
  683.19      .1       0
#XS Ineff= 1 ,-1
  329.76  928.59 2501.09
Permanent Ineff=
       F
Bank Sta=274.36,294.42
XS Rating Curve= 0 ,0
Exp/Cntr=0.3,0.1

Type RM Length L Ch R = 1 ,9042    ,323.4,328.4,333.2
XS GIS Cut Line= 4
2140606.08418439401506.3076141482140249.09638131401445.543956146
2139981.08445014401509.5628569722139630.60680464401512.818099812
#Sta/Elev= 30
       0 2624.48    20.5  2615.6    30.5 2609.64    37.1 2608.51    80.4 2589.83
   143.6 2559.25   200.2 2536.68   240.2 2526.38   276.8 2522.18   342.7 2501.18
   393.7 2495.58     397 2494.59   409.8 2486.01  438.592486.372   447.1 2485.17
  457.252486.813   467.9 2489.59   538.7 2488.88   556.9 2490.63   592.7 2489.03
     668 2500.88   695.6 2511.62     737 2535.65   762.2 2548.29   814.2 2583.46
     896 2632.88   939.1 2653.73   948.3 2659.33   964.7 2662.74   988.2 2675.58
#Mann= 5 ,-1 , 0
       0      .1       0   61.83      .1       0  438.59    .045       0
  457.25      .1       0  759.35      .1       0
#XS Ineff= 1 ,-1
  468.02  988.16  2494.6
Permanent Ineff=
       F
Bank Sta=438.59,457.25
XS Rating Curve= 0 ,0
Exp/Cntr=0.3,0.1

Type RM Length L Ch R = 1 ,8714    ,296.1,312.8,316.3
XS GIS Cut Line= 3
2140583.29781264401326.186255232 2139943.1068358401182.957210973
2139625.18161863  401127.6184109
#Sta/Elev= 30
       0 2591.22     7.5 2589.79    54.5 2567.07     115 2542.23     152  2535.9
   289.2 2523.93     310 2516.85   320.5 2508.48   333.6 2505.63   350.7 2496.29
   390.7 2485.38   404.2 2483.43   447.9 2482.28   466.1 2483.86   538.6 2482.09
   552.1 2479.66   568.9 2479.08  574.682476.689   582.3 2474.85  594.832475.709
   602.5 2477.58   676.3 2532.16   723.8 2549.26   766.1    2567   806.2 2589.61
     887 2638.57   929.4 2660.34   939.4 2666.85   952.7 2670.34   978.7 2684.44
#Mann= 5 ,-1 , 0
       0      .1       0   45.51      .1       0  553.33      .1       0
  574.68    .045       0  594.83      .1       0
Bank Sta=574.68,594.83
XS Rating Curve= 0 ,0
Exp/Cntr=0.3,0.1

Type RM Length L Ch R = 1 ,8401    ,254.8,240.7,230.9
XS GIS Cut Line= 4
2140437.89849713401150.4051107322140199.18342339401019.111738145
2139948.53234988400842.2452939752139706.56170522400741.333750397
#Sta/Elev= 30
       0    2543    44.6  2539.1    85.7 2533.74   161.3 2528.12     285 2514.19
   301.1  2506.1   333.2 2484.33   341.3 2480.43   365.3 2478.24   381.4 2478.43
   397.5 2470.97   405.5 2468.89   425.6 2471.11   441.6 2470.25   445.42468.329
   457.7 2466.77  484.922467.986   489.8 2469.81   499.2 2479.19   516.3  2489.9
     530 2494.79   545.5 2503.35   585.9 2522.14   603.2 2528.68   635.2 2537.73
   649.4 2543.59   721.4 2581.02   748.9 2593.47   798.7 2608.25   841.4 2616.57
#Mann= 4 ,-1 , 0
       0      .1       0  151.74      .1       0   445.4    .045       0
  484.92      .1       0
#XS Ineff= 2 , 0
          432.37 2475.08
Permanent Ineff=
       F       F
Bank Sta=445.4,484.92
XS Rating Curve= 0 ,0
Exp/Cntr=0.3,0.1

Type RM Length L Ch R = 1 ,8160    ,255,261.7,267.6
XS GIS Cut Line= 4
2140570.27716939400740.2487788052140191.58796614 400687.08024998
 2139952.8725643400700.1012213082139728.26310539400659.953663811
#Sta/Elev= 30
       0 2560.32   113.5 2522.34   143.3  2517.9   186.4 2516.65   269.2 2505.64
   295.7 2494.97   328.8 2478.67   335.4 2478.61     352 2482.44   361.9 2487.02
   391.7 2487.15     395 2486.31   414.7 2471.51   424.5 2462.22     441 2459.63
   467.3  2458.2  475.182460.089   480.4 2463.56   496.8 2465.37   519.8 2472.33
   529.7 2478.48   562.5 2503.15   611.8  2525.3   670.3 2542.48   708.5 2551.84
     725 2558.05   741.7 2559.92   758.3 2564.04   815.7 2581.31   849.6 2593.06
#Mann= 3 , 0 , 0
       0      .1       0     441    .045       0  475.18      .1       0
Bank Sta=441,475.18
XS Rating Curve= 0 ,0
Exp/Cntr=0.3,0.1

Type RM Length L Ch R = 1 ,7898    ,200.8,201.2,201
XS GIS Cut Line= 2
2140627.78558455400690.3354928052139923.57570688400327.922503725
#Sta/Elev= 30
       0 2590.76    32.4 2582.34    95.1 2562.45   222.7 2509.47   246.4 2501.53
   251.9 2500.43   322.6 2494.55   331.3 2491.97   359.1 2479.49   368.9 2476.13
   382.9 2474.12   408.7  2473.4   427.3 2470.11     442    2469   456.7 2462.97
   489.9 2458.16     515 2458.53   523.1 2456.29   534.2 2450.16  537.922448.917
   551.6 2448.43  557.962448.541   566.2 2449.66   571.1 2452.11   585.7 2468.78
   607.6 2484.23   696.5 2527.82   744.5 2557.73   770.3 2571.52     792 2588.43
#Mann= 3 ,-1 , 0
       0      .1       0  537.92    .045       0  557.96      .1       0
Bank Sta=537.92,557.96
XS Rating Curve= 0 ,0
Exp/Cntr=0.3,0.1

Type RM Length L Ch R = 1 ,7697    ,244.3,244.1,243.1
XS GIS Cut Line= 2
2140641.89152747400476.5767339772140004.95579347400142.375630721
#Sta/Elev= 30
       0 2573.25    47.5 2546.71   115.1 2513.75   148.5  2500.5   186.1  2488.6
   233.7 2476.37   289.3 2473.21   326.3 2462.89   396.7  2455.5   422.7 2457.12
   429.1 2455.05   443.6 2446.44  452.48 2443.02   462.4 2442.59  472.592443.884
   480.1 2444.96   493.1 2442.83   507.9 2447.24   518.9 2448.68   545.7 2460.47
   559.7 2464.44   572.4 2465.51   589.4 2472.37   608.9 2488.05   626.4 2503.64
   641.3 2514.55     655 2527.51   685.7  2552.2   693.1 2560.77   719.3  2582.3
#Mann= 5 ,-1 , 0
       0      .1       0   105.4     .05       0  353.83      .1       0
  452.48    .045       0  472.59      .1       0
Bank Sta=452.48,472.59
XS Rating Curve= 0 ,0
Exp/Cntr=0.3,0.1

Type RM Length L Ch R = 1 ,7453    ,193.1,190.8,188.3
XS GIS Cut Line= 2
2140735.20761381400233.5214458112140085.25090846399941.637515143
#Sta/Elev= 30
       0 2579.07    19.8 2566.99    59.4 2545.01   127.7 2509.05   156.5 2494.98
   195.9 2477.56   215.7 2471.19     268 2461.64   290.2 2459.82     304 2457.63
   329.1 2449.92   347.1 2446.22   375.9 2444.84   433.4  2446.4   444.1 2443.64
     455 2443.31   466.4 2439.83   483.8 2439.63  502.972437.352   512.6 2437.03
  523.052438.505   537.7 2441.56   552.1 2448.33   566.5 2451.69   577.3 2456.32
   595.5 2467.18     642 2500.58   669.9 2513.56   688.8 2519.26   712.5 2528.84
#Mann= 5 ,-1 , 0
       0      .1       0  389.96    .055       0  435.27      .1       0
  502.97    .045       0  523.05      .1       0
Bank Sta=502.97,523.05
XS Rating Curve= 0 ,0
Exp/Cntr=0.3,0.1

Type RM Length L Ch R = 1 ,7262    ,243.5,253,262.4
XS GIS Cut Line= 3
2140813.90729576400045.0615176012140538.16932079399881.150610262
2140130.68986891399807.620483605
#Sta/Elev= 30
       0 2574.61    65.8 2540.45   116.4 2517.93   135.5 2511.59   211.9 2491.45
   221.4 2487.77     231 2487.08   268.6 2476.17   276.7  2474.7   295.8 2466.62
   325.6 2449.77   332.3 2447.17   365.7 2441.54     379 2437.22   401.2 2439.35
   425.7 2436.61     509 2436.17   528.62432.018     539 2431.87   548.62432.614
     569 2434.96     579 2434.16     589 2435.94   598.9  2440.5   642.4 2464.57
     659 2475.84   675.7 2484.92   708.8 2497.16   722.4 2499.94   734.8 2499.85
#Mann= 5 ,-1 , 0
       0      .1       0   268.6    .055       0   425.7      .1       0
   528.6    .045       0   548.6      .1       0
#XS Ineff= 2 , 0
          508.96 2436.68
Permanent Ineff=
       F       F
Bank Sta=528.6,548.6
XS Rating Curve= 0 ,0
Exp/Cntr(USF)=0,0
Exp/Cntr=0.5,0.3

Type RM Length L Ch R = 1 ,7009    ,53.7,54.7,55.4
XS GIS Cut Line= 5
 2140817.8716419400014.0664245872140459.06346591399699.481105021
 2140436.9520377399649.2278590842140405.79502522399587.918899041
2140148.49840602399422.083187449
#Sta/Elev= 30
       0 2567.18    82.2 2531.92   151.9 2508.99   176.8 2499.83   191.7  2491.6
   202.8 2489.72   221.5  2481.6   260.6 2470.16   291.1 2467.15   352.2 2455.33
   360.9 2451.06   370.2 2441.08   377.2 2437.12   391.1 2436.08   400.7 2432.16
   425.6 2431.46   451.6 2431.65   541.22426.657   562.7 2426.15   563.6 2426.14
   605.2 2429.77   663.8 2450.71   695.5 2450.39   714.2 2446.34   730.8 2447.42
     745 2440.68   753.5 2439.81     777  2452.8   819.9 2463.07     907 2495.29
#Mann= 5 ,-1 , 0
       0      .1       0   425.6    .055       0   451.6      .1       0
   541.2    .045       0   562.7      .1       0
#XS Ineff= 3 ,-1
       0   521.2  2428.9   582.7  584.31  2428.9  584.31     800 2433.92
Permanent Ineff=
       F       F       F
Bank Sta=541.2,562.7
XS Rating Curve= 0 ,0
Exp/Cntr(USF)=0,0
Exp/Cntr=0.5,0.3

Type RM Length L Ch R = 1 ,6955    ,162.7,156,147
XS GIS Cut Line= 4
2140837.97294027399998.9904508062140502.28125742399682.395001403
2140449.01281672399548.7213672112140189.70606769399385.900850375
#Sta/Elev= 30
       0 2572.38    37.9 2555.37    90.5 2535.54   138.3 2511.21   197.7 2505.07
   211.2 2496.08   229.2 2494.37   251.8 2482.82   296.1 2467.74   312.8 2459.62
   324.8 2455.96     342  2445.5     351 2442.12   436.7 2428.88   454.3 2431.54
   473.5 2431.11   487.7  2428.2   528.1 2428.55   546.12424.869   554.8 2424.69
   567.22425.226   612.4 2427.82   633.6 2425.28   671.9 2426.87   699.4 2429.93
   732.9 2436.36   755.2 2435.41   774.2 2431.39   807.9 2448.14   911.5 2479.05
#Mann= 3 ,-1 , 0
       0      .1       0   546.1    .045       0   567.2      .1       0
#XS Ineff= 2 , 0
                          614.04         2432.26
Permanent Ineff=
       F       F
Bank Sta=546.1,567.2
XS Rating Curve= 0 ,0
Exp/Cntr(USF)=0,0
Exp/Cntr=0.5,0.3

Type RM Length L Ch R = 1 ,6799    ,373.1,378.3,381.5
XS GIS Cut Line= 3
2140928.34994406399615.0318691432140510.59815489399464.207039565
2140219.79952389399360.040253147
#Sta/Elev= 30
       0 2612.62    36.2 2588.34    60.7 2569.56    85.1 2554.97    98.1 2542.84
     106 2540.38     116 2534.04   126.3  2531.3   137.4 2522.26   154.8 2512.16
   224.6 2478.11   290.9 2448.66   297.8 2445.02   315.3  2431.4   325.8 2429.17
   336.4 2422.82   357.1 2421.81   362.52420.126  379.482419.709   416.4 2420.71
   454.8 2418.55   468.7 2418.94   479.2    2425   548.9 2421.82   632.5 2422.32
   646.5 2427.08   660.4 2437.57   677.8 2446.43   726.6 2459.96     753 2469.19
#Mann= 3 ,-1 , 0
       0      .1       0   362.5    .045       0  379.48      .1       0
#XS Ineff= 2 , 0
          354.12 2430.79  481.27          2435.8
Permanent Ineff=
       F       F
Bank Sta=362.5,379.48
XS Rating Curve= 0 ,0
Exp/Cntr=0.3,0.1

Type RM Length L Ch R = 1 ,6420    ,258.2,245.3,236.8
XS GIS Cut Line= 3
2140998.87933056399325.3182097232140366.28413905399067.071678981
2140159.03586589398996.542292476
#Sta/Elev= 30
       0 2593.86      35 2572.63     113 2536.76   127.2 2532.53   144.6 2520.72
   180.3 2505.58   247.7 2489.01   311.4 2469.22   343.3 2452.96     361 2439.73
   371.7  2437.3   389.4  2424.2   407.1 2414.73   449.6 2411.81   460.3 2408.32
     478 2411.32  506.74 2406.27   529.6 2404.68  536.162406.175   548.9  2411.2
   591.4 2406.08   615.2 2416.35   626.8 2417.11   644.5 2427.32   712.5 2445.68
   773.6 2452.38   801.4 2450.47   815.2 2455.95   884.8 2463.04   902.2 2467.84
#Mann= 3 ,-1 , 0
       0      .1       0  506.74    .045       0  536.16      .1       0
#XS Ineff= 2 , 0
          478.78 2417.59  559.71         2418.84
Permanent Ineff=
       F       F
Bank Sta=506.74,536.16
XS Rating Curve= 0 ,0
Exp/Cntr=0.3,0.1

Type RM Length L Ch R = 1 ,6175    ,230.4,228.5,226.9
XS GIS Cut Line= 4
2140960.90204431398850.0576773142140708.08069955398855.483191401
2140442.23871155398924.9276063142140181.82223764 398963.99019222
#Sta/Elev= 30
       0 2529.01      24 2528.12    53.5 2531.02    72.6 2530.93    99.5 2528.42
   120.9 2522.96   149.7 2511.32   243.9 2463.82   284.8 2436.07   311.7 2413.86
   322.4 2402.88   375.8 2405.18   392.8 2403.44  403.342400.469   432.7 2398.83
  441.752399.905     464 2400.04   497.9 2416.68   511.4 2417.86   518.2 2422.86
     525 2424.97     558 2426.48   571.5 2423.37   614.6 2435.76   661.1 2444.33
   690.9 2448.82   704.2  2448.7   714.2 2452.03   747.3 2452.72     791 2467.36
#Mann= 5 ,-1 , 0
       0      .1       0  226.37      .1       0  314.38      .1       0
  403.34    .045       0  441.75      .1       0
#XS Ineff= 2 , 0
          361.74 2410.35
Permanent Ineff=
       F       F
Bank Sta=403.34,441.75
XS Rating Curve= 0 ,0
Exp/Cntr=0.3,0.1

Type RM Length L Ch R = 1 ,5946    ,224.8,226.4,227.5
XS GIS Cut Line= 3
2140791.63105738398552.7488887312140397.75093964398714.424090311
2140142.75965172398822.931091145
#Sta/Elev= 30
       0 2479.31    27.4 2471.47    48.6 2466.68    62.8  2466.4   119.6 2459.78
   165.7 2448.64   205.2 2442.42   211.8 2440.49   220.3 2436.29   247.2 2417.19
   275.6  2401.5   286.3 2400.27   311.1 2393.47   332.82393.278   348.5 2392.79
  352.872393.208   368.6 2394.79   383.7 2397.93   411.4 2397.64   463.8 2399.72
   474.5 2401.71   491.5 2407.94   513.7 2409.92     524 2412.29   556.5 2416.18
   581.4 2420.42   617.1 2432.64     632  2441.6   671.6 2461.07   702.9 2477.96
#Mann= 4 ,-1 , 0
       0      .1       0   332.8    .045       0  352.87      .1       0
  402.73      .1       0
Bank Sta=332.8,352.87
XS Rating Curve= 0 ,0
Exp/Cntr=0.3,0.1

Type RM Length L Ch R = 1 ,5720    ,243.9,223.9,210.4
XS GIS Cut Line= 3
2140639.72158431398411.6897876412140361.94359656398480.049230978
2139997.36033621398583.130717725
#Sta/Elev= 30
       0 2450.27    72.4 2444.46    94.6 2440.66   133.2 2435.92   158.1    2431
   160.2  2429.8   173.7 2414.46   190.6 2402.32   204.1 2389.56  208.05 2387.04
   214.3 2385.19   224.4 2385.12   237.3 2386.87   244.7 2388.46   264.9 2388.74
   275.1 2390.91   304.1 2389.84   325.4  2387.7   363.6 2390.12   377.3 2389.13
   397.7 2390.45   414.8 2397.11   459.1 2394.43   492.9  2395.4   503.8 2396.98
   516.8 2400.75   534.1 2408.94     639    2469     650 2473.23   664.9 2484.56
#Mann= 5 ,-1 , 0
       0      .1       0    94.6      .1       0  208.05    .045       0
   237.3      .1       0   304.1      .1       0
#XS Ineff= 2 , 0
                          278.89         2394.32
Permanent Ineff=
       F       F
Bank Sta=208.05,237.3
XS Rating Curve= 0 ,0
Exp/Cntr=0.5,0.3

Type RM Length L Ch R = 1 ,5496    ,54.9,55.4,54.2
XS GIS Cut Line= 5
2140569.53596243398148.5328187022140251.86946104398250.477369293
2140245.49792663398366.0752079092140227.29354259398425.239456019
2140047.07014066398552.670144257
#Sta/Elev= 30
       0  2468.9    65.5 2451.29     162 2422.88   183.6 2414.17   213.7 2397.85
   220.6 2395.67   226.5 2394.92   237.8 2395.63   248.2 2394.54   265.4 2396.77
   275.7  2396.9     282 2394.64   296.4 2384.09   299.8 2382.96     353 2383.54
   373.1 2381.61   399.4 2380.59   415.9 2380.19   424.6 2381.11   445.4 2384.52
   476.1 2386.36   519.5 2386.76   561.1 2392.81   614.6  2393.7   634.7 2397.14
   642.7 2399.78   658.8 2407.39   698.3 2430.51   707.8 2435.15     732 2450.83
#Mann= 3 ,-1 , 0
       0      .1       0   399.4    .045       0   424.6      .1       0
#XS Ineff= 2 , 0
           389.4  2381.3   434.6          2381.3
Permanent Ineff=
       F       F
Bank Sta=399.4,424.6
XS Rating Curve= 0 ,0
Exp/Cntr(USF)=0,0
Exp/Cntr=0.5,0.3

Type RM Length L Ch R = 1 ,5441    ,319.8,342,363.1
XS GIS Cut Line= 6
2140554.97245521 398142.16128429 2140232.7548578398201.325532401
2140199.98696654398234.0934236622140199.98696654398348.781043076
2140193.61543213 398404.30441438 2140016.1226878398559.041678669
#Sta/Elev= 30
       0 2465.24    78.7 2442.56     112 2430.88   152.1 2419.72   178.7 2409.59
   202.4 2399.26   232.1  2391.4   244.1 2390.57     261 2387.99   282.1 2382.79
   289.2 2381.74   429.8 2379.03   439.6 2378.01   449.5 2378.27     454 2379.59
   459.3 2382.14   472.4 2384.17   525.2 2386.64   544.5 2389.13   568.2 2389.17
   585.2 2391.97   622.7 2393.11   636.6 2394.72   650.1 2397.57     664 2402.61
   680.7 2411.72   698.8 2420.21   720.3    2433   754.9 2455.45     780  2469.4
#Mann= 3 ,-1 , 0
       0      .1       0   429.8    .045       0     454      .1       0
#XS Ineff= 2 , 0
          339.86 2386.42
Permanent Ineff=
       F       F
Bank Sta=429.8,454
XS Rating Curve= 0 ,0
Exp/Cntr(USF)=0,0
Exp/Cntr=0.5,0.3

Type RM Length L Ch R = 1 ,5099    ,308.8,311.4,314.5
XS GIS Cut Line= 2
2140565.93662688398137.167042732 2139912.7250068 397885.43099764
#Sta/Elev= 30
       0 2468.42      63  2450.7    94.7    2439   111.5 2430.57     143 2412.79
   201.4 2385.81   217.7 2379.23   229.3 2377.33   249.6 2376.45   316.2 2376.43
   337.3 2374.42   354.9 2375.82     383 2374.96   414.6 2372.63  421.89 2369.78
   425.2 2368.57   434.9 2368.15   442.8 2368.31  451.432370.339   460.3 2374.07
   489.1  2392.8   523.7 2421.95   542.3 2432.85     577 2459.01     608 2476.91
   625.3 2483.99   653.7 2498.21   674.8    2512   686.2 2517.29     700    2526
#Mann= 5 ,-1 , 0
       0      .1       0     1.2      .1       0  388.26      .1       0
  421.89    .045       0  451.43      .1       0
#XS Ineff= 2 , 0
          368.53 2381.26
Permanent Ineff=
       F       F
Bank Sta=421.89,451.43
XS Rating Curve= 0 ,0
Exp/Cntr=0.3,0.1

Type RM Length L Ch R = 1 ,4787    ,422.3,424.7,408.2
XS GIS Cut Line= 2
2140686.37962747397978.7470839772140137.33446573397591.377123818
#Sta/Elev= 30
       0 2500.92    54.8 2474.99    94.9 2454.69   150.2 2430.51   167.2 2421.55
   183.2 2411.27   195.3 2404.93   216.1 2390.69     249 2371.48   274.9 2368.56
   319.7 2366.03   382.2 2366.44   393.5 2364.23   409.1 2368.34   428.2 2363.21
   440.2 2363.21   452.3 2364.96  474.642363.667  495.012362.909     496  2362.9
   500.4 2363.39   504.5 2366.05   516.5 2378.25   522.1 2383.01   536.3 2393.95
   552.7 2408.11   580.7 2429.39   616.9 2454.33   649.6 2474.72   671.9  2487.6
#Mann= 7 ,-1 , 0
       0      .1       0  261.89      .1       0  322.39      .1       0
  371.25      .1       0  451.43      .1       0  474.64    .045       0
  495.01      .1       0
#XS Ineff= 2 , 0
          411.21 2373.47
Permanent Ineff=
       F       F
Bank Sta=474.64,495.01
XS Rating Curve= 0 ,0
Exp/Cntr=0.3,0.1

Type RM Length L Ch R = 1 ,4363    ,487.7,484.4,467.1
XS GIS Cut Line= 3
2140931.60518689397641.2904098032140590.89326988397478.529908568
2140309.86036739397377.618364975
#Sta/Elev= 30
       0  2520.3    15.9 2511.13    33.6 2502.57   143.2 2440.95   161.4 2432.36
   186.8 2417.83   215.9 2402.77   267.4 2371.69     285 2362.61   295.9 2362.03
   299.1 2360.78  304.54 2355.37   306.8 2353.96   310.4 2353.78  338.532355.618
   350.4 2356.59   370.7 2352.96   393.4 2357.62   424.3 2355.37   449.2 2357.03
   457.7 2356.34   466.6 2354.08     498 2355.38     509 2361.23   557.2 2394.92
   617.2 2429.62   646.3 2444.66   657.7 2449.34   665.4 2451.76   676.2 2452.35
#Mann= 5 ,-1 , 0
       0      .1       0  304.54    .045       0  338.53      .1       0
  415.88      .1       0  593.24      .1       0
Bank Sta=304.54,338.53
XS Rating Curve= 0 ,0
Exp/Cntr=0.3,0.1

Type RM Length L Ch R = 1 ,3878    ,284.1,282.3,281.1
XS GIS Cut Line= 2
2141072.66428797397015.2053758952140316.37085305397123.712376729
#Sta/Elev= 30
       0 2517.51    60.9 2477.72    84.1 2459.77    97.4 2452.72   123.9 2434.59
   173.7 2402.88   223.3 2367.34   243.2  2357.7   266.4 2351.34     283 2348.68
   326.1 2346.68   342.6 2346.72   358.9 2348.56   372.5 2346.32     389 2347.69
   438.8 2344.81  449.242341.063   455.3 2339.78   468.6 2339.89  476.192341.659
   481.8 2344.58   491.8 2346.51   511.7  2346.5   521.6 2345.25   528.2 2346.99
   584.6 2390.65   597.8 2398.58   617.7 2408.56   712.8 2426.88     764 2438.85
#Mann= 3 ,-1 , 0
       0      .1       0  449.24    .045       0  476.19      .1       0
#XS Ineff= 2 , 0
                          497.57         2355.59
Permanent Ineff=
       F       F
Bank Sta=449.24,476.19
XS Rating Curve= 0 ,0
Exp/Cntr=0.3,0.1

Type RM Length L Ch R = 1 ,3596    ,430.1,431.5,432.2
XS GIS Cut Line= 2
2140952.22161546396698.3651303052140281.64848155396878.486489221
#Sta/Elev= 30
       0 2480.25    26.2 2462.21    46.4    2450    76.9 2426.09   104.2 2415.99
   141.5  2392.1   195.9 2363.27   202.7 2357.81   212.9 2353.03   219.7 2347.46
   246.9 2345.73   259.1 2340.41   287.6 2336.55   328.4 2337.15   389.5 2340.19
  419.232334.988   433.2 2332.84   447.3 2333.19  451.982334.626   460.9 2338.98
   471.1 2340.68     505 2359.61   525.4 2367.12   552.6 2371.98   576.4 2370.94
   600.2 2366.97   606.9 2367.46   634.3  2375.7   674.9 2395.75   694.3 2403.25
#Mann= 5 ,-1 , 0
       0      .1       0  207.71      .1       0  296.05      .1       0
  419.23    .045       0  451.98      .1       0
#XS Ineff= 2 , 0
          385.06 2352.11
Permanent Ineff=
       F       F
Bank Sta=419.23,451.98
XS Rating Curve= 0 ,0
Exp/Cntr=0.3,0.1
